HEC-RAS study BigClearCk.prj: BigClearCk

--- BigClearCk.g01 (geometry) --- (continued)

Type RM Length L Ch R = 1 ,56171.1 ,466.3,397.8,455.2
XS GIS Cut Line= 2
     2079273.582       384242.94     2078894.384      384641.576
#Sta/Elev= 30
       0 3168.49      20 3161.47      40 3154.25     100  3131.8     110 3127.94
     130 3119.76   180.1 3098.48   190.1 3095.19   200.1 3093.45   230.1 3092.05
   240.1 3091.16   250.1 3089.39   260.1  3087.1   270.1  3084.4   280.1 3081.94
   290.1 3081.08   295.1 3081.51   300.1 3081.94   310.1 3085.08   320.1 3088.49
   330.1 3091.49   390.1 3107.76   400.1 3110.63   420.1 3116.78   480.2 3136.75
   490.2 3140.19   500.2 3143.86   510.2 3147.72   520.2 3151.74   550.2 3164.37
#Mann= 3 , 0 , 0
       0      .1       0   280.1    .045       0   295.1      .1       0
Bank Sta=280.1,295.1
XS Rating Curve= 0 ,0
Exp/Cntr=0.3,0.1

Type RM Length L Ch R = 1 ,55773.1 ,348.9,363.5,378.1
XS GIS Cut Line= 2
     2078930.001      383976.984     2078602.143      384446.572
#Sta/Elev= 30
       0 3157.78    30.1 3147.37    50.2 3140.71    90.4  3128.3   100.5 3124.92
   110.5 3121.17   120.6 3116.94   150.7 3103.75   180.9 3091.94     201 3083.38
     211 3079.97     221 3077.37   241.1 3072.79   261.2 3067.56   264.9 3067.04
   271.3 3066.13   279.9 3066.48   281.3 3066.54   291.4 3068.79   301.4    3072
   311.5 3074.98   351.7 3085.67     432 3101.83   492.3 3113.72   502.4 3115.93
   512.4 3118.71   522.5 3121.87   532.5 3125.38   552.6 3133.16   572.7  3141.7
#Mann= 3 , 0 , 0
       0      .1       0   264.9    .045       0   279.9      .1       0
Bank Sta=264.9,279.9
XS Rating Curve= 0 ,0
Exp/Cntr=0.3,0.1

Type RM Length L Ch R = 1 ,55409.7 ,375.7,376.2,376.3
XS GIS Cut Line= 2
     2078846.157       383879.24     2078286.539      384088.574
#Sta/Elev= 30
       0 3143.23    49.8 3126.94    69.7 3120.02    89.6 3112.65   119.5 3102.99
   129.5 3099.06   139.4 3094.63   149.4 3090.68   179.2 3080.97   189.2 3078.11
   199.2 3076.21   219.1  3074.1   278.8 3064.81   298.7 3062.29   368.4 3056.81
   405.9 3054.61   418.2 3054.49   420.9 3054.91   428.2 3056.05   438.2 3059.74
   458.1 3069.28     488 3082.02   507.9 3090.82   537.7 3104.81   547.7 3109.86
   557.7 3115.78   567.6 3123.12   577.6 3131.36   587.5 3140.46   597.5  3150.5
#Mann= 3 , 0 , 0
       0      .1       0   405.9    .045       0   420.9      .1       0
Bank Sta=405.9,420.9
XS Rating Curve= 0 ,0
Exp/Cntr=0.3,0.1

Type RM Length L Ch R = 1 ,55033.2 ,323.4,323.4,323.4
XS GIS Cut Line= 2
     2078798.196      383576.879     2078182.472        383807.2
#Sta/Elev= 30
       0 3137.35    59.8 3116.18   109.6 3097.54   159.4 3077.09   209.2 3054.54
   219.1 3054.17     239 3061.62     249 3063.56     259 3062.97   278.9 3056.74
   298.8  3048.3   308.8 3045.17   312.7 3044.86   318.7 3044.38   327.7 3044.96
   378.5 3049.66   398.4 3053.26   408.4 3056.72   468.1 3082.36   478.1 3085.71
   488.1 3087.37     508  3088.9   527.9  3092.9   537.9 3096.59   557.8 3106.62
   607.6 3140.12   627.5 3152.06   637.5 3155.12   647.4 3154.09   657.4 3150.34
#Mann= 3 , 0 , 0
       0      .1       0   312.7    .045       0   327.7      .1       0
Bank Sta=312.7,327.7
XS Rating Curve= 0 ,0
Exp/Cntr=0.3,0.1

Type RM Length L Ch R = 1 ,54709.8 ,249.9,255.2,260.6
XS GIS Cut Line= 2
     2078746.726      383252.392     2078105.244      383492.348
#Sta/Elev= 30
       0 3128.89    80.6 3095.35   151.1 3064.58   181.3 3051.76   201.4 3044.06
   221.6 3037.29   231.6 3035.93   241.7 3037.73   251.8 3041.18     282  3050.6
   292.1 3052.38   302.2 3051.84   312.2 3049.42   322.3 3046.26   342.4 3039.07
   352.8 3036.08   362.6 3035.29   367.8  3036.3   372.7 3037.25   392.8  3045.7
     423  3057.2   433.1 3060.24   453.2 3063.18   463.3 3065.78   473.4 3069.29
   513.7 3084.27     564 3103.38   664.8 3142.71   674.8 3146.48   684.9 3149.71
#Mann= 3 , 0 , 0
       0      .1       0   352.8    .045       0   367.8      .1       0
#XS Ineff= 2 , 0
          298.85 3051.98
Permanent Ineff=
       F       F
Bank Sta=352.8,367.8
XS Rating Curve= 0 ,0
Exp/Cntr=0.3,0.1

Type RM Length L Ch R = 1 ,54454.3 ,277.6,277.6,277.7
XS GIS Cut Line= 2
     2078720.278      383085.656      2078026.63      383171.842
#Sta/Elev= 30
       0 3136.71    89.9  3105.5   169.8 3076.42   189.7 3066.34   219.7 3046.24
   229.7 3040.79   239.6 3036.26   249.6 3033.05   259.6 3030.96   269.6 3030.04
   279.6 3030.72   289.6 3033.76   309.6 3043.64   319.5 3045.28   329.5  3043.4
   339.5 3039.29   359.5 3028.93   369.5 3024.78   374.1 3023.99   379.4 3023.07
   389.1 3023.45   399.4 3025.33   439.4 3038.24   449.4 3040.37   479.3 3042.34
   529.2 3048.58   619.1 3065.65   639.1 3067.23     649 3066.63     699 3060.67
#Mann= 3 , 0 , 0
       0      .1       0   374.1    .045       0   389.1      .1       0
#XS Ineff= 2 , 0
          319.93 3045.13
Permanent Ineff=
       F       F
Bank Sta=374.1,389.1
XS Rating Curve= 0 ,0
Exp/Cntr=0.3,0.1

Type RM Length L Ch R = 1 ,54176.8 ,329.4,335.4,341.3
XS GIS Cut Line= 2
     2078677.968      382818.922      2077982.29      382905.359
#Sta/Elev= 30
       0 3161.74    60.1 3136.68   150.2 3103.33   220.3 3076.42   260.4    3060
   280.4 3051.39   300.4 3042.33   310.5 3039.22   320.5 3036.79   330.5 3032.66
   340.5 3027.37   350.5 3023.19   360.5 3021.58   380.6 3021.81   390.6 3021.16
   400.6 3019.89   420.6  3015.7   427.4 3014.69   430.6 3014.22   440.6 3014.05
   442.4 3014.28   450.7 3015.32   480.7 3021.22   490.7 3022.36   510.8 3023.58
   520.8 3025.13   530.8 3027.16     651 3053.78     671 3058.69     701  3067.2
#Mann= 3 , 0 , 0
       0      .1       0   427.4    .045       0   442.4      .1       0
Bank Sta=427.4,442.4
XS Rating Curve= 0 ,0
Exp/Cntr=0.3,0.1

Type RM Length L Ch R = 1 ,53840.5 ,309.3,303.2,297
XS GIS Cut Line= 2
     2078643.873      382603.971     2077931.244      382499.676
#Sta/Elev= 30
       0 3130.14      20 3122.87     120 3087.73   180.1 3064.29   200.1 3056.85
   240.1 3043.16   270.1  3033.5   280.1 3030.86   300.1 3026.52   320.1 3019.42
   330.1 3016.45   340.1 3014.08   350.1 3012.52   419.1 3005.67   430.1  3005.4
   434.1 3005.74   440.1 3006.26   460.1 3009.95   510.2 3017.81   530.2 3019.16
   540.2 3020.46   610.2 3038.46   630.2 3043.06   640.2 3044.63   650.2 3045.52
   660.2 3045.92   670.2  3046.9   680.2 3048.91   700.2 3054.43   720.2 3060.71
#Mann= 3 , 0 , 0
       0      .1       0   419.1    .045       0   434.1      .1       0
Bank Sta=419.1,434.1
XS Rating Curve= 0 ,0
Exp/Cntr=0.3,0.1

Type RM Length L Ch R = 1 ,53537.2 ,467.2,478.7,490.2
XS GIS Cut Line= 2
     2078582.346      382216.084     2077906.132      382300.103
#Sta/Elev= 30
       0 3120.55      20 3112.72    30.1 3108.63    40.1 3104.38    50.1 3099.92
   120.2 3067.47   210.4 3026.77   220.5 3022.78   230.5 3020.25   240.5 3017.89
   250.5 3013.84   270.6 3002.87   280.6  2999.4   285.2 2998.88   290.6 2998.27
   300.2 2998.38   360.8 3001.48     471 3007.54     491 3008.41     501 3009.09
   511.1 3011.42   521.1  3015.8   531.1 3020.71   561.2 3034.48   571.2 3039.15
   591.2 3048.63   611.3 3058.43   631.3 3068.71   651.4 3079.35   681.4 3095.85
#Mann= 3 , 0 , 0
       0      .1       0   285.2    .045       0   300.2      .1       0
Bank Sta=285.2,300.2
XS Rating Curve= 0 ,0
Exp/Cntr=0.3,0.1

Type RM Length L Ch R = 1 ,53056.8 ,407.5,408.1,408.7
XS GIS Cut Line= 2
      2078507.42      381979.251      2077972.18      381768.349
#Sta/Elev= 30
       0 3068.99    10.1 3062.26    20.2  3056.3    30.3  3050.8    40.4 3045.49
    50.5 3040.53   100.9  3014.7     111 3010.58   121.1 3008.54   141.3 3008.18
   151.4 3007.32   171.6 3004.65     222 3001.31   282.6 2995.34   312.9 2992.74
   333.1 2991.24   373.4 2988.96   405.1  2988.6   413.8 2988.32   420.1 2988.43
   423.9  2988.5     434 2991.03   454.2 3001.66   464.3 3004.46   474.4 3006.23
   484.5  3010.3   514.7 3029.19   534.9 3042.75   565.2 3063.75   575.3 3070.23
#Mann= 3 , 0 , 0
       0      .1       0   405.1    .045       0   420.1      .1       0
Bank Sta=405.1,420.1
XS Rating Curve= 0 ,0
Exp/Cntr=0.3,0.1

Type RM Length L Ch R = 1 ,52649   ,291.9,294.2,296.4
XS GIS Cut Line= 2
     2078627.733      381679.523     2078098.504      381453.089
#Sta/Elev= 30
       0 3061.84     9.9 3056.82    29.8 3045.85    49.6 3033.55    69.5 3022.13
    79.4 3017.08    89.3 3012.57   109.2 3004.73   119.1 3001.54     129 2999.25
     139 2998.03   148.9 2996.26   158.8 2992.94   168.7 2989.05   188.6 2979.66
   199.4  2976.7   208.4 2976.24   214.4 2976.41     268 2977.82   287.8 2979.17
   297.7 2980.54   347.4 2989.32     397 2998.99   416.8  3001.9   426.8 3002.94
   446.6 3004.12   456.5 3005.86   496.2 3020.04   516.1 3028.06   575.6 3050.03
#Mann= 3 , 0 , 0
       0      .1       0   199.4    .045       0   214.4      .1       0
Bank Sta=199.4,214.4
XS Rating Curve= 0 ,0
Exp/Cntr=0.3,0.1

Type RM Length L Ch R = 1 ,52354.2 ,374.5,371.8,369.1
XS GIS Cut Line= 2
     2078725.505      381435.951     2078218.711      381153.093
#Sta/Elev= 30
       0 3015.12      10 3011.88      20 3008.86      30 3006.08      40  3003.6
      50 3001.26      60 2999.08    90.1    2993   110.1 2989.98   120.1  2987.5
   130.1 2983.98   140.1  2979.3   150.1 2973.87   160.1 2970.76   170.1 2969.93
   174.2 2970.07   180.1 2970.26   189.2  2970.9   200.1 2971.73   240.2 2974.45
   340.2 2983.43   380.2  2987.2   390.3 2987.85   400.3 2988.75   410.3  2991.2
   420.3 2995.58   430.3 3000.45   490.3 3030.17   520.4 3045.32   580.4 3075.82
#Mann= 3 , 0 , 0
       0      .1       0   174.2    .045       0   189.2      .1       0
Bank Sta=174.2,189.2
XS Rating Curve= 0 ,0
Exp/Cntr=0.3,0.1

Type RM Length L Ch R = 1 ,51982.4 ,411.8,392.4,373.1
XS GIS Cut Line= 2
     2078865.505       381087.18     2078335.915      380860.592
#Sta/Elev= 30
       0    3000    69.5 2983.23    79.4 2981.02    89.4 2979.52   109.2  2977.9
   188.7  2969.2   218.5 2965.51   238.4 2962.46   248.3 2961.62   252.5 2961.69
   258.2 2961.79   267.5 2962.91   278.1 2964.71     288 2966.27   307.9 2968.88
   317.8 2969.55   327.7 2970.39   337.7 2972.53   357.5 2978.36   377.4 2984.03
     427 2999.42     437 3003.23   446.9 3008.22   456.8  3012.8   466.8 3016.23
   496.6 3025.09   516.4  3031.2   526.4 3034.37   556.2 3044.06     576 3050.29
#Mann= 3 , 0 , 0
       0      .1       0   252.5    .045       0   267.5      .1       0
Bank Sta=252.5,267.5
XS Rating Curve= 0 ,0
Exp/Cntr=0.3,0.1

Type RM Length L Ch R = 1 ,51589.9 ,315.9,311.7,307.4
XS GIS Cut Line= 2
     2078955.075      380486.078     2078369.516      380760.423
#Sta/Elev= 30
       0 3066.06    19.9 3059.05    59.7 3045.82    79.6 3038.88   109.4 3027.87
   119.4 3023.32   129.3 3017.54   139.3 3010.82   159.2 2996.65   208.9 2960.14
   218.9 2954.15   228.8 2952.89   238.8 2956.13   248.7    2960   258.7 2961.36
   268.6  2960.1   278.6 2957.28   298.4  2950.2   308.5 2948.27   318.4 2947.96
   323.5 2948.26   417.8 2955.57   507.4 2957.77   517.3 2958.52   527.3 2960.68
   537.2 2964.66   557.1 2974.58   606.8 3000.08   626.7 3009.64   646.6 3018.59
#Mann= 3 , 0 , 0
       0      .1       0   308.5    .045       0   323.5      .1       0
#XS Ineff= 2 , 0
          257.93 2961.32
Permanent Ineff=
       F       F
Bank Sta=308.5,323.5
XS Rating Curve= 0 ,0
Exp/Cntr=0.3,0.1

Type RM Length L Ch R = 1 ,51278.5 ,379.9,383.1,386.4
XS GIS Cut Line= 2
     2078790.289      380156.507      2078253.77      380541.115
#Sta/Elev= 30
       0    3058      70 3036.38     110 3023.33     120 3020.46     130 3018.72
     140 3017.42     150 3014.53     160 3008.92     170 3001.23     210 2969.26
     240 2944.97     250 2940.06     260 2940.49   280.1 2949.66   290.1 2951.08
   300.1 2950.62   310.1 2949.46   350.1 2944.24   373.1 2940.66   380.1 2939.82
   388.1 2939.99   420.1 2943.22   430.1 2943.94   510.1 2945.84   540.1 2947.22
   550.1 2948.42   560.1 2951.36   570.1 2955.98   590.1 2966.52   660.1 3005.81
#Mann= 3 , 0 , 0
       0      .1       0   373.1    .045       0   388.1      .1       0
#XS Ineff= 2 , 0
          292.65 2951.09
Permanent Ineff=
       F       F
Bank Sta=373.1,388.1
XS Rating Curve= 0 ,0
Exp/Cntr=0.3,0.1

Type RM Length L Ch R = 1 ,50895   ,314.1,309.6,305.2
XS GIS Cut Line= 2
     2078649.611      379875.151     2078058.378      380170.899
#Sta/Elev= 30
       0 3009.55      30 3002.21    80.1 2994.07    90.2 2991.85   100.2  2988.8
   260.4 2930.54   270.4 2929.79   280.5 2933.44   290.5 2938.95   300.5 2942.09
   310.5 2941.82   320.5 2939.99   360.6 2930.13   364.7 2929.74   370.6 2929.18
   379.7 2929.86   410.7 2936.62   440.7 2938.79   460.8 2942.34   480.8 2947.69
   500.8 2955.26   510.8 2960.61   520.8 2968.06   530.9  2977.2   540.9 2985.25
   550.9 2991.09   570.9 3001.38     581 3007.41     631 3042.63   661.1 3060.25
#Mann= 3 , 0 , 0
       0      .1       0   364.7    .045       0   379.7      .1       0
#XS Ineff= 2 , 0
          301.95 2942.13
Permanent Ineff=
       F       F
Bank Sta=364.7,379.7
XS Rating Curve= 0 ,0
Exp/Cntr=0.3,0.1

Type RM Length L Ch R = 1 ,50585.4 ,408.2,398.8,389.3
XS GIS Cut Line= 2
     2078476.758      379529.445     2077926.575      379969.524
#Sta/Elev= 30
       0 2995.39    70.4 2973.32   100.6 2963.45   191.2 2937.62   261.7 2918.91
   271.8 2916.94   281.8 2916.49   291.9 2918.51     312 2925.88   322.1 2928.85
   332.1 2929.89   342.2 2928.31   362.3 2920.58   372.1 2917.62   382.5  2916.9
   387.1 2917.76   392.5 2918.76   402.6    2922   412.7 2924.52   432.8    2927
     473 2937.24   483.1 2940.77   493.2 2944.97   583.8 2985.85   593.8 2989.74
   603.9 2992.99   644.2 3004.29   664.3 3010.44   684.4 3017.41   704.5 3025.14
#Mann= 3 , 0 , 0
       0      .1       0   372.1    .045       0   387.1      .1       0
#XS Ineff= 2 , 0
          331.62 2929.67
Permanent Ineff=
       F       F
Bank Sta=372.1,387.1
XS Rating Curve= 0 ,0
Exp/Cntr=0.3,0.1

Type RM Length L Ch R = 1 ,50186.6 ,251.6,249.8,247.9
XS GIS Cut Line= 2
     2077971.368      379333.836     2077775.348      379710.698
#Sta/Elev= 26
       0 2982.52    29.6 2969.69    59.3 2956.97    88.9 2944.13    98.8 2939.92
   118.6 2931.73   138.3 2923.44   148.2 2920.02   167.9 2915.19   177.8 2911.66
   187.7 2907.28   197.6 2904.29     202 2903.95   207.5 2903.53     217  2904.2
   256.8 2909.23   266.7 2910.28   286.5 2911.42   296.4 2912.52   306.2 2914.15
   335.9 2919.67   345.8 2921.89   355.6 2925.17   365.5 2928.99   395.2 2940.69
   424.8 2952.46
#Mann= 3 , 0 , 0
       0      .1       0     202    .045       0     217      .1       0
Bank Sta=202,217
XS Rating Curve= 0 ,0
Exp/Cntr=0.3,0.1

Type RM Length L Ch R = 1 ,49936.8 ,229.2,229.2,229.2
XS GIS Cut Line= 2
     2077694.419      379304.951     2077565.305      379611.474
#Sta/Elev= 30
       0 2957.53    10.1 2951.49    20.2 2944.92    40.3  2931.1    50.4 2924.58
    60.5 2918.68    70.6 2913.99    80.6 2911.29    90.7 2909.19   100.8 2906.26
   110.9  2902.6     121 2899.29   122.9    2899     131 2897.74   137.9 2897.95
   141.1 2898.05   151.2 2899.47   181.4 2904.26   191.5 2905.34   201.6 2905.88
   211.7 2906.72   221.7 2908.34   241.9 2912.01     252 2914.21     262 2917.28
   272.1 2921.01   302.4 2932.65   312.4 2935.74   322.5  2937.2   332.6  2937.2
#Mann= 3 , 0 , 0
       0      .1       0   122.9    .045       0   137.9      .1       0
Bank Sta=122.9,137.9
XS Rating Curve= 0 ,0
Exp/Cntr=0.3,0.1

Type RM Length L Ch R = 1 ,49707.6 ,252,252,252
XS GIS Cut Line= 2
     2077484.819      379213.298     2077358.291      379513.683
#Sta/Elev= 29
       0 2933.85     9.9 2928.04    19.8 2922.43    29.6 2917.32    39.5 2912.97
    49.4 2909.28    59.3 2906.32    69.1 2904.47      79 2903.41    88.9 2902.59
    98.8 2901.29   108.6 2899.37   118.5 2897.09   128.4 2894.64   137.6 2892.71
   138.3 2892.56   148.2 2891.96   152.6  2892.4     158 2892.93   177.8 2896.79
   187.7  2898.5   197.5 2899.74   217.3 2901.28   227.2 2902.78   266.7 2911.34
   276.6 2913.35   286.4 2915.18   306.2 2918.63     326 2921.82
#Mann= 3 , 0 , 0
       0      .1       0   137.6    .045       0   152.6      .1       0
Bank Sta=137.6,152.6
XS Rating Curve= 0 ,0
Exp/Cntr=0.3,0.1

Type RM Length L Ch R = 1 ,49455.6 ,297,298,299.1
XS GIS Cut Line= 2
     2077254.289      379112.493     2077114.337      379444.746
#Sta/Elev= 30
       0 2924.47      20 2917.53      30 2914.17    80.1 2897.87    90.1 2895.67
   100.2 2894.28   110.2 2892.68   120.2 2890.48   130.2 2887.79   140.2 2885.21
   148.5 2884.19   150.2 2883.98   160.2 2884.74   163.5 2885.43   170.2 2886.84
   180.3 2888.26   190.3 2888.74   200.3 2888.81   210.3  2889.2   220.3 2889.97
   240.4 2892.31   250.4 2893.92   260.4 2896.35   270.4 2899.37   280.4 2903.17
   290.4 2908.21   300.4 2914.01   310.4 2919.34   320.5 2924.09   360.5 2941.79
#Mann= 3 , 0 , 0
       0      .1       0   148.5    .045       0   163.5      .1       0
Bank Sta=148.5,163.5
XS Rating Curve= 0 ,0
Exp/Cntr=0.3,0.1

Type RM Length L Ch R = 1 ,49157.1 ,309.5,319.2,328.9
XS GIS Cut Line= 2
     2076990.552      378997.167     2076816.858      379362.731
#Sta/Elev= 30
       0 2894.91     9.9 2893.27    29.6 2889.77    39.5 2888.83    49.4 2888.53
   128.3 2887.46   138.2 2886.97   148.1  2885.6   157.9 2883.08   167.8 2880.01
   174.3 2878.39   177.7 2877.55   187.6 2876.96   189.3 2877.05   197.4  2877.5
   207.3 2878.33   217.2 2879.31     227 2880.85   246.8  2884.5   256.7 2887.41
   266.5 2893.77   276.4 2902.86   286.3 2910.84   296.1 2916.74     306 2921.79
   315.9 2926.68   325.8 2931.54   335.6 2936.17     385 2958.23   404.7 2967.26
#Mann= 3 , 0 , 0
       0      .1       0   174.3    .045       0   189.3      .1       0
Bank Sta=174.3,189.3
XS Rating Curve= 0 ,0
Exp/Cntr=0.3,0.1

Type RM Length L Ch R = 1 ,48837.9 ,216.3,222.3,228.3
XS GIS Cut Line= 2
     2076807.269      378868.213     2076533.682      379096.797
#Sta/Elev= 20
       0 2881.73    79.2 2882.59   128.7 2882.97   158.4 2883.29   168.4 2882.89
   178.3    2881   188.2 2877.92   198.1 2873.99     208 2870.99   209.4 2870.84
   217.9  2869.9   224.4 2870.45   227.8 2870.74   237.7 2872.84   247.6 2874.61
   257.5 2875.72   267.4 2877.73   277.3 2881.64   316.9 2901.73   356.5 2921.54
#Mann= 3 , 0 , 0
       0      .1       0   209.4    .045       0   224.4      .1       0
Bank Sta=209.4,224.4
XS Rating Curve= 0 ,0
Exp/Cntr=0.3,0.1

Type RM Length L Ch R = 1 ,48615.5 ,286,302.3,318.7
XS GIS Cut Line= 2
     2076752.183      378721.712      2076383.68      378890.545
#Sta/Elev= 21
       0 2876.25    29.7 2876.62   138.4 2878.22   197.7 2878.79   217.5 2878.79
   227.4 2877.97   237.3 2875.82   247.2 2872.38     257 2868.48   266.9 2865.89
   271.5 2865.82   276.8 2865.75   286.5 2867.34   296.6 2870.27   306.5 2872.23
   316.4 2873.08   326.2 2874.13   336.1 2875.79     346 2877.69   375.7 2882.85
   405.3 2887.76
#Mann= 3 , 0 , 0
       0      .1       0   271.5    .045       0   286.5      .1       0
Bank Sta=271.5,286.5
XS Rating Curve= 0 ,0
Exp/Cntr=0.3,0.1

Type RM Length L Ch R = 1 ,48312.8 ,247.5,249.9,252.3
XS GIS Cut Line= 2
     2076686.207      378636.842     2076302.556      378522.515
#Sta/Elev= 22
       0 2874.76    70.1 2873.71   120.1 2872.65   150.1 2871.89   180.2 2870.96
   220.2 2869.29   230.2 2868.72   240.2  2867.6   250.2 2865.82   270.2 2860.95
   274.2 2860.37   280.2  2859.5   289.2 2859.38   290.2 2859.37   300.2 2860.89
   310.2 2863.72   320.3 2866.03   330.3 2867.43   340.3 2869.95   350.3 2874.87
   370.3 2887.08   400.3 2905.88
#Mann= 3 , 0 , 0
       0      .1       0   274.2    .045       0   289.2      .1       0
Bank Sta=274.2,289.2
XS Rating Curve= 0 ,0
Exp/Cntr=0.3,0.1

Type RM Length L Ch R = 1 ,48063.1 ,263,246.4,229.9
XS GIS Cut Line= 2
     2076695.596      378406.606     2076344.143      378256.962
#Sta/Elev= 30
       0 2868.02    20.1  2867.1    30.2 2866.55    60.3 2864.69    80.4  2863.6
   100.5  2862.9   130.7 2862.37   140.7 2861.92   150.8 2860.72   160.8 2858.98
   170.9  2857.1   180.9  2854.9     191 2852.56   192.6 2852.32     201 2851.09
   207.6 2851.19   211.1 2851.25   221.2 2852.47   231.2 2854.26   241.2 2855.56
   251.3 2856.54   261.4 2857.36   271.4 2858.05   281.5 2858.56   301.6 2859.15
   321.7 2859.45   331.7 2859.86   361.9 2862.04   371.9 2863.32     382 2865.75
#Mann= 3 , 0 , 0
       0      .1       0   192.6    .045       0   207.6      .1       0
Bank Sta=192.6,207.6
XS Rating Curve= 0 ,0
Exp/Cntr=0.3,0.1

Type RM Length L Ch R = 1 ,47816.6 ,292.6,292.6,292.7
XS GIS Cut Line= 2
     2076768.666      378035.015     2076344.143      378177.425
#Sta/Elev= 30
       0 2909.74      10 2906.06    19.9  2902.2    59.7 2886.13    79.6 2878.31
    89.6  2874.2    99.5 2869.79   109.5 2865.72   119.4    2863   129.4 2861.29
   139.3 2860.07   149.3 2859.06   159.2 2857.42   169.2 2855.06   179.1 2852.43
     199 2846.84   205.5 2845.74     209 2845.14   218.9 2845.24   220.5 2845.56
   228.9 2847.22   238.8  2850.3   248.8 2852.26   258.7 2852.94   328.4 2854.34
   378.1 2854.82     408 2855.43   417.9 2855.82   427.9  2856.6   447.8 2858.55
#Mann= 3 , 0 , 0
       0      .1       0   205.5    .045       0   220.5      .1       0
Bank Sta=205.5,220.5
XS Rating Curve= 0 ,0
Exp/Cntr=0.3,0.1

Type RM Length L Ch R = 1 ,47523.8 ,361.6,358.9,356.2
XS GIS Cut Line= 2
     2076717.699      377747.746     2076284.099      377893.201
#Sta/Elev= 30
       0 2884.16    29.8 2876.83    79.5 2865.59   109.4 2859.28   139.2  2853.5
   149.1 2851.89   159.1 2850.96     169 2850.34     179 2849.41   188.9 2848.15
   218.7 2844.14   238.6 2841.64   258.5 2838.65   268.4 2836.77   278.9 2835.27
   288.3  2834.8   293.9 2835.08   298.3  2835.3   308.2 2836.86   318.2 2838.76
   328.1 2840.16     338 2841.07   377.8 2844.24   387.8 2844.87   397.7 2845.23
   407.6 2846.48   417.6  2848.8   437.5 2854.26   447.4 2857.46   457.4 2861.02
#Mann= 3 , 0 , 0
       0      .1       0   278.9    .045       0   293.9      .1       0
Bank Sta=278.9,293.9
XS Rating Curve= 0 ,0
Exp/Cntr=0.3,0.1

Type RM Length L Ch R = 1 ,47164.8 ,347.3,347.3,347.3
XS GIS Cut Line= 2
     2076591.151      377401.252     2076145.417      377615.838
#Sta/Elev= 30
       0 2856.93    10.1 2854.98    60.6 2843.08    80.8  2838.7    90.9 2836.75
     101 2835.87     111 2836.22   121.2  2837.3   141.3 2839.85   151.4 2840.51
   161.5 2840.24   171.6 2839.06     212 2833.08   222.1 2830.89   232.2 2827.89
   237.3 2826.89   242.3  2825.9   252.3 2825.67   272.6 2826.92   292.8  2827.4
   302.9 2828.02   363.4 2832.72   383.6 2833.92   393.7  2835.5   403.8  2840.2
   413.9 2847.84     424 2856.55   464.4  2892.8   484.6 2907.34   494.7 2912.58
#Mann= 3 , 0 , 0
       0      .1       0   237.3    .045       0   252.3      .1       0
Bank Sta=237.3,252.3
XS Rating Curve= 0 ,0
Exp/Cntr=0.3,0.1

Type RM Length L Ch R = 1 ,46817.4 ,417.2,412.9,408.7
XS GIS Cut Line= 2
     2076435.074      377139.794     2075952.833      377371.956
#Sta/Elev= 30
       0 2852.19    49.6 2844.33    59.5  2842.5   138.8 2826.52   148.7  2824.7
   158.6 2823.58   168.5 2823.97   178.4 2825.01     218 2830.37     228  2831.3
   237.9 2831.31   247.8  2830.7   257.7  2829.7   287.4  2826.1   346.9  2818.2
   369.8  2814.4   376.6 2813.59   384.8  2813.5   386.5 2813.48   396.5 2815.17
   416.3 2823.26   426.2 2826.02   436.1 2827.66     446 2829.64   455.9 2834.37
   465.8 2842.08   495.6 2867.52   515.4 2883.96   525.3  2891.7   535.2 2897.46
#Mann= 3 , 0 , 0
       0      .1       0   369.8    .045       0   384.8      .1       0
Bank Sta=369.8,384.8
XS Rating Curve= 0 ,0
Exp/Cntr=0.3,0.1

Type RM Length L Ch R = 1 ,46404.5 ,339.7,338,336.7
XS GIS Cut Line= 2
     2076165.302      376782.189     2075724.206      377101.131
#Sta/Elev= 30
       0 2840.29    20.2  2836.4    30.2 2834.75    70.6 2828.44   191.5 2808.07
   211.7 2803.84   221.8 2802.59   222.8 2802.61   231.8 2802.76   237.8 2803.43
     252 2804.98   282.2 2807.43   292.3 2808.34   302.4 2809.52   362.9 2818.08
     373 2819.43     383 2820.42   393.1 2820.61   423.4 2820.86   433.4 2821.32
   443.5 2822.46   453.6 2823.94   463.7 2825.76   473.8 2827.91   483.8  2830.4
   493.9 2833.32     504 2836.62   514.1 2840.25   534.2 2847.71   544.3  2851.3
#Mann= 3 , 0 , 0
       0      .1       0   222.8    .045       0   237.8      .1       0
Bank Sta=222.8,237.8
XS Rating Curve= 0 ,0
Exp/Cntr=0.3,0.1

Type RM Length L Ch R = 1 ,46066.5 ,398.5,365.4,411.9
XS GIS Cut Line= 2
     2076030.277      376444.943     2075478.923      376900.403
#Sta/Elev= 30
       0 2895.65    20.1 2885.74    40.3 2876.85    60.4 2869.94    80.6 2865.41
   130.9 2856.52   161.2 2847.96   171.2 2845.76   201.4 2841.16   221.6 2837.33
   231.7 2834.59     282 2815.47   312.2  2805.6   332.4 2798.25   342.5 2795.04
   352.5 2794.16   354.2 2794.23   362.6 2794.56   369.2 2795.36   453.3 2805.52
   493.6  2809.7   543.9 2811.84     554 2812.03   594.3 2811.18   604.4 2811.92
   614.4 2814.43   664.8  2830.5   674.9 2832.69   684.9 2833.42   715.2 2833.79
#Mann= 3 , 0 , 0
       0      .1       0   354.2    .045       0   369.2      .1       0
Bank Sta=354.2,369.2
XS Rating Curve= 0 ,0
Exp/Cntr=0.3,0.1

Type RM Length L Ch R = 1 ,45701.1 ,318.3,318.3,318.3
XS GIS Cut Line= 2
      2075795.92      376248.023     2075325.322      376505.764
#Sta/Elev= 30
       0 2878.61     9.9 2874.08    69.6 2848.21   109.3 2830.84   119.2 2826.98
   129.2 2823.94   139.1 2821.87   168.9 2815.99   188.8 2811.73   228.5 2802.69
   268.3 2793.39   288.2 2788.22   295.6 2786.93   298.1  2786.5     308 2786.24
   310.6 2786.45     318 2787.06   367.6 2793.99   377.6 2795.15   387.5 2795.84
   397.4 2796.23   407.4 2796.86   427.3 2798.78   437.2 2799.24   457.1 2799.16
   496.8 2798.35   506.8 2798.03   516.7 2797.55   526.6 2797.31   536.6 2797.46
#Mann= 3 , 0 , 0
       0      .1       0   295.6    .045       0   310.6      .1       0
Bank Sta=295.6,310.6
XS Rating Curve= 0 ,0
Exp/Cntr=0.3,0.1

Type RM Length L Ch R = 1 ,45382.8 ,319.5,319.6,319.7
XS GIS Cut Line= 2
     2075647.194      375974.053     2075145.301      376248.934
#Sta/Elev= 30
       0 2884.42    40.2 2867.37    50.2 2862.69    70.3 2852.59    80.3 2847.74
   110.4 2834.22   180.7 2803.26   200.8 2794.57   210.8 2789.97   220.9 2784.66
   230.9 2780.41   237.3 2779.38   240.9  2778.8   252.3 2779.33   271.1 2781.08
   311.2 2784.12   361.4 2787.71   371.4 2788.26   391.5 2788.83   411.6 2790.23
   421.6 2790.67   431.7 2790.66   441.7 2790.44   471.8 2789.56   491.9 2788.78
     512 2787.76     522 2787.91   532.1 2788.25   562.2  2788.4   572.2 2788.74
#Mann= 3 , 0 , 0
       0      .1       0   237.3    .045       0   252.3      .1       0
Bank Sta=237.3,252.3
XS Rating Curve= 0 ,0
Exp/Cntr=0.3,0.1

Type RM Length L Ch R = 1 ,45063.2 ,242.4,246,249.5
XS GIS Cut Line= 2
      2075496.07      375695.667     2074962.378      375987.963
#Sta/Elev= 30
       0 2864.38    29.9 2853.06    69.8 2838.84    79.8 2835.08    89.8 2830.85
    99.8 2826.19   109.7    2821   139.6 2804.55   159.6 2794.12   169.6 2789.28
   179.6  2784.9   189.5 2781.23   199.5 2778.76   209.5 2777.56   219.5  2776.9
   274.5 2776.07   279.3 2776.03   289.5 2776.46   349.1 2780.73   379.1 2781.76
     409 2783.37     419 2783.25   448.9 2781.33   458.9 2781.45   478.8 2782.54
   508.7  2783.5   518.7 2784.52   528.7 2786.54   548.6  2791.7   608.5 2805.61
#Mann= 3 , 0 , 0
       0      .1       0   274.5    .045       0   289.5      .1       0
Bank Sta=274.5,289.5
XS Rating Curve= 0 ,0
Exp/Cntr=0.3,0.1

Type RM Length L Ch R = 1 ,44817.2 ,207.6,208.8,210
XS GIS Cut Line= 2
     2075404.477      375526.944     2074832.124       375728.94
#Sta/Elev= 30
       0  2839.8    79.6  2813.9    99.5 2806.84   139.3    2792   149.2 2788.42
   159.2 2785.09     189 2775.65     199 2772.84     209 2771.08   218.9  2770.5
   248.8 2770.22   306.9 2768.54   308.4  2768.5   318.4  2768.7   321.9 2769.06
   328.4 2769.72   348.2  2772.4   378.1 2775.67     388 2776.62     398 2777.12
   467.6 2777.79   507.4 2777.52   517.4  2778.3   527.4 2780.45   537.3 2783.55
   547.2 2787.04   567.2 2794.41   577.1 2797.83     587 2801.18     607 2807.39
#Mann= 3 , 0 , 0
       0      .1       0   306.9    .045       0   321.9      .1       0
Bank Sta=306.9,321.9
XS Rating Curve= 0 ,0
Exp/Cntr=0.3,0.1

Type RM Length L Ch R = 1 ,44608.3 ,187.4,199.3,211.2
XS GIS Cut Line= 2
     2075326.956       375349.79     2074746.487      375521.116
#Sta/Elev= 30
       0 2813.77    40.4 2798.74    50.4 2795.33    60.5  2792.4    70.6 2789.78
     111 2779.57     121 2777.43   131.1 2776.11   141.2 2775.33   191.6 2772.14
   211.8 2770.58   282.4 2763.96   295.1 2762.98   302.6 2762.76   310.1 2763.12
   312.7 2763.25   332.9 2765.63     353  2767.6   373.2 2768.79   413.6 2769.53
   494.3 2771.84   504.4 2772.02   524.5 2771.98   534.6  2772.4   544.7 2774.46
   554.8 2778.35   564.9 2783.56     575 2789.56     585 2795.12   605.2 2805.44
#Mann= 3 , 0 , 0
       0      .1       0   295.1    .045       0   310.1      .1       0
Bank Sta=295.1,310.1
XS Rating Curve= 0 ,0
Exp/Cntr=0.3,0.1

Type RM Length L Ch R = 1 ,44408.9 ,305.4,304.9,304.5
XS GIS Cut Line= 2
     2075334.087      375316.922     2074743.895      375182.867
#Sta/Elev= 30
       0 2816.22    50.4 2796.31    60.5 2792.76    70.6 2789.88    80.7  2787.5
   131.1 2776.25   141.2 2774.39   151.3 2773.06   161.4 2772.08   322.8 2757.56
   337.8 2756.47     343 2756.26   352.8 2756.75   383.3 2761.69   393.4  2762.2
   413.6 2761.59   423.7 2761.78   433.7 2762.65   453.9 2765.33     464 2766.97
   474.1 2769.36   484.2 2773.34   494.3  2779.1   514.4 2792.48   524.5 2798.41
   534.6 2803.49   544.7 2807.69   554.8 2811.13     575 2816.64   605.2 2826.09
#Mann= 3 , 0 , 0
       0      .1       0   337.8    .045       0   352.8      .1       0
Bank Sta=337.8,352.8
XS Rating Curve= 0 ,0
Exp/Cntr=0.3,0.1

Type RM Length L Ch R = 1 ,44104   ,360.2,352.7,345.3
XS GIS Cut Line= 2
      2075425.65      375030.652     2074835.458      374896.597
#Sta/Elev= 30
       0 2831.08    10.1 2826.52    40.4 2812.33    50.4 2808.47    60.5 2805.58
   161.4 2780.83   181.6 2776.07     232 2765.57   242.1 2763.66   272.4 2759.16
   292.5 2756.57     343  2751.9   370.1 2749.15   373.2 2748.86   383.3 2748.68
   385.1 2748.87   393.4 2749.74   413.6 2753.66   423.7 2755.45   433.7 2757.14
   443.8 2758.58   453.9 2759.44   474.1 2759.78   484.2 2760.35   494.3 2762.16
   504.4    2765   554.8 2780.44     585 2789.33   595.1 2792.69   605.2  2796.3
#Mann= 3 , 0 , 0
       0      .1       0   370.1    .045       0   385.1      .1       0
Bank Sta=370.1,385.1
XS Rating Curve= 0 ,0
Exp/Cntr=0.3,0.1

Type RM Length L Ch R = 1 ,43751.3 ,301.7,295.7,289.7
XS GIS Cut Line= 2
      2075498.15      374580.045     2074801.269      374656.667
#Sta/Elev= 30
       0 2857.78    60.1 2840.91    70.1 2837.91    80.1 2834.66   100.2 2827.47
   150.2 2809.16   170.3 2802.16   220.3 2784.12   270.4 2766.43   290.4 2759.76
   320.5 2750.15   340.5 2742.91   350.3 2740.97   360.6 2740.86   365.3 2741.39
   370.6 2741.99   390.6 2745.02   450.7 2753.39   460.7 2754.61   470.7 2754.76
   480.7 2754.02   490.8 2753.54   500.8 2753.72   510.8 2755.16   520.8 2757.84
   540.8 2764.32   610.9 2788.13     631 2794.72     661    2805   701.1  2818.3
#Mann= 3 , 0 , 0
       0      .1       0   350.3    .045       0   365.3      .1       0
Bank Sta=350.3,365.3
XS Rating Curve= 0 ,0
Exp/Cntr=0.3,0.1

Type RM Length L Ch R = 1 ,43455.6 ,302.1,302.1,302.1
XS GIS Cut Line= 2
     2075378.611       374221.43     2074762.606      374463.352
#Sta/Elev= 30
       0 2820.48    80.2  2800.3   100.3 2795.01   120.3 2789.42   140.4 2783.28
   180.5  2770.7   200.6 2763.88   250.7 2744.95   260.7 2740.79   270.7 2736.27
   278.2 2733.75   280.8 2732.88   290.8 2732.07   293.2 2732.29   300.8    2733
   330.9  2737.9     371 2743.69   401.1 2748.95   411.1 2750.24   431.2 2751.22
   441.2  2752.4   461.3 2755.69   471.3 2757.69   491.3 2762.26   531.4 2772.38
   621.7 2793.13   631.7 2796.01   641.8 2799.97   651.8 2804.86   661.8 2810.14
#Mann= 3 , 0 , 0
       0      .1       0   278.2    .045       0   293.2      .1       0
Bank Sta=278.2,293.2
XS Rating Curve= 0 ,0
Exp/Cntr=0.3,0.1

Type RM Length L Ch R = 1 ,43153.5 ,402.3,404.3,406.4
XS GIS Cut Line= 2
     2075287.789      373934.793     2074702.839      374164.518
#Sta/Elev= 30
       0 2805.54    69.8 2789.95    79.8  2787.1   109.7 2777.03   119.7 2774.01
   129.7 2771.59   209.5 2757.18   229.4 2753.09   239.4 2750.27   249.4 2746.93
   279.3 2736.42   299.3 2728.89   309.2 2725.94   317.5 2725.18   319.2 2725.03
   329.2 2725.56   332.5 2726.01     409 2736.74   438.9  2741.9   448.9 2743.27
   468.8 2744.75   478.8 2747.01   488.8 2750.89   498.8 2755.53   518.7 2765.68
   538.7 2777.05   558.6 2789.17   588.5 2806.52   608.5 2816.76   628.4 2825.54
#Mann= 3 , 0 , 0
       0      .1       0   317.5    .045       0   332.5      .1       0
Bank Sta=317.5,332.5
XS Rating Curve= 0 ,0
Exp/Cntr=0.3,0.1

Type RM Length L Ch R = 1 ,42749.2 ,463,465.2,467.5
XS GIS Cut Line= 2
     2075131.524      373608.648     2074533.644      373782.408
#Sta/Elev= 30
       0 2778.67    30.1  2769.6    40.2 2766.91    60.2 2762.78   100.4 2755.72
   261.1 2728.74   291.2 2724.81   350.6 2718.14   361.5  2717.3   365.6 2717.34
   371.6  2717.4   381.6 2719.36   401.7 2726.17   411.7  2728.9   421.8 2730.81
   431.8 2731.77   451.9 2732.45   461.9 2733.22     472 2736.77     482 2743.04
   502.1 2757.11   512.2 2763.35   522.2 2768.93   532.2 2773.63   542.3 2777.45
   552.3 2780.66   562.4 2783.28   602.5 2791.12   612.6 2793.54   622.6 2796.36
#Mann= 3 , 0 , 0
       0      .1       0   350.6    .045       0   365.6      .1       0
Bank Sta=350.6,365.6
XS Rating Curve= 0 ,0
Exp/Cntr=0.3,0.1

Type RM Length L Ch R = 1 ,42284   ,383.1,380.9,378.6
XS GIS Cut Line= 2
      2075085.02      373184.931     2074496.818      373293.947
#Sta/Elev= 30
       0 2815.92      10 2811.06    19.9 2805.57    49.8 2787.36    59.8 2781.66
    69.8 2776.51    79.8 2771.88    99.7 2763.23   119.6 2753.88   129.6 2749.89
   139.6 2746.92   259.2 2717.37   269.2 2715.32   279.2 2714.05   289.1 2713.45
   385.8 2709.54   388.8 2709.48   398.8 2709.97   400.8 2710.27   438.7 2716.37
   468.6 2722.24   478.6 2723.43   498.5 2724.31   508.5  2725.6   528.4  2729.2
   538.4 2731.58   548.4 2734.34   558.3 2737.38   578.3 2743.98   598.2 2750.93
#Mann= 3 , 0 , 0
       0      .1       0   385.8    .045       0   400.8      .1       0
Bank Sta=385.8,400.8
XS Rating Curve= 0 ,0
Exp/Cntr=0.3,0.1

Type RM Length L Ch R = 1 ,41903.1 ,421.5,434.4,447.3
XS GIS Cut Line= 2
     2074978.212      372781.853      2074434.69      372939.816
#Sta/Elev= 30
       0 2775.15    29.8 2765.73    39.7 2762.11    59.6  2753.9    79.4 2745.58
    89.4 2741.61    99.3 2738.26   109.2  2735.7   158.9 2724.71   198.6 2715.68
   208.5 2713.52   218.5  2711.9   228.4 2710.91   268.1 2708.51   337.6 2704.55
   359.8 2703.07   367.4 2702.71   374.8  2703.1   377.3 2703.23   387.3 2705.01
   397.2 2707.18   407.1 2709.16   417.1 2710.87     427 2712.05   436.9 2712.64
   456.8 2713.15   466.7 2714.18   476.6 2716.59   486.6 2719.92     566 2748.03
#Mann= 3 , 0 , 0
       0      .1       0   359.8    .045       0   374.8      .1       0
Bank Sta=359.8,374.8
XS Rating Curve= 0 ,0
Exp/Cntr=0.3,0.1

Type RM Length L Ch R = 1 ,41468.7 ,544,532.2,517.9
XS GIS Cut Line= 2
     2075060.963      372587.387      2074281.12      372359.801
#Sta/Elev= 30
       0 2793.63    50.2 2772.51   140.4 2732.86   150.4 2729.24   160.5 2726.26
   240.7 2705.31   250.7 2703.77   260.8 2703.35   300.9 2702.92     351 2700.94
   371.1 2699.39   411.2 2694.85   440.8 2692.17   441.3 2692.14   455.8 2692.52
   471.4 2694.48   511.5 2701.22   531.6 2702.72   551.6 2702.63   581.7 2699.84
   591.7 2699.42   621.8 2702.05   641.9 2702.82     672 2704.95   712.1 2702.89
   732.1 2703.28   742.2 2705.22   752.2 2709.09   772.3 2720.41   812.4 2745.62
#Mann= 3 , 0 , 0
       0      .1       0   440.8    .045       0   455.8      .1       0
Bank Sta=440.8,455.8
XS Rating Curve= 0 ,0
Exp/Cntr=0.3,0.1

Type RM Length L Ch R = 1 ,40936.3 ,299.6,288.2,276.9
XS GIS Cut Line= 2
     2075462.957      371783.139     2074367.553      372106.458
#Sta/Elev= 30
       0 2698.18    50.1 2698.93   130.2 2695.86   190.4 2694.97   260.5 2695.17
   310.6 2696.69   360.7 2693.39   410.8 2692.81   440.8 2693.86   500.9 2698.86
     521 2699.92     551 2697.56   591.1 2697.99   671.2 2695.31   681.3  2693.5
   701.3 2688.74   721.3 2685.95   736.2 2684.85   741.4 2684.77   751.2 2684.77
   771.4 2685.02   791.5 2686.45   801.5 2687.67   831.6 2693.08   841.6 2693.91
  1001.9 2691.43    1062 2691.23    1082 2691.99  1122.1 2697.22  1142.1 2697.56
#Mann= 3 , 0 , 0
       0     .06       0   736.2    .045       0   751.2      .1       0
#XS Ineff= 2 , 0
          519.75  2699.9  850.31         2693.97
Permanent Ineff=
       F       F
Bank Sta=736.2,751.2
XS Rating Curve= 0 ,0
Exp/Cntr=0.3,0.1

Type RM Length L Ch R = 1 ,40648.1 ,265.3,265.2,265.2
XS GIS Cut Line= 2
     2075300.471      371212.801     2074374.716      372059.255
#Sta/Elev= 30
       0 2763.56    40.1 2757.32    70.2 2755.74    90.3 2753.68   180.6 2739.46
   250.9 2729.56     271 2727.86   311.1 2727.14   351.2 2723.92   371.3 2721.59
   421.5 2713.61   491.7 2709.08   541.9 2702.68   612.1 2697.32   652.3 2695.14
   692.4 2693.78   702.5 2692.74   712.5 2690.61   732.6 2684.84   742.6 2683.59
   752.6 2683.41   760.9 2683.45   775.9 2684.24   812.8 2689.54   832.9  2690.8
   913.2 2690.32  1043.7 2691.21  1204.2 2689.78  1214.2 2690.52  1254.4 2696.93
#Mann= 3 , 0 , 0
       0     .06       0   760.9    .045       0   775.9     .06       0
#XS Ineff= 2 , 0
                         1049.07         2691.17
Permanent Ineff=
       F       F
Bank Sta=760.9,775.9
XS Rating Curve= 0 ,0
Exp/Cntr=0.3,0.1

Type RM Length L Ch R = 1 ,40382.9 ,782.3,764.5,746.6
XS GIS Cut Line= 2
     2074970.938      371156.296     2074126.621      371928.287
#Sta/Elev= 30
       0 2795.51    30.1 2788.84    80.3 2776.05   140.5 2763.86   160.6 2759.11
   200.7  2746.8   240.8 2732.45   250.9 2730.33   260.9 2729.18   331.2 2724.99
   341.2 2723.41   351.2  2720.5   411.5 2697.18   421.5 2693.72   431.5 2691.28
   511.8 2682.01     547 2681.67     552 2681.63     562 2681.71   622.2 2684.97
   732.6 2686.93     833 2686.99   963.4 2684.93   973.4 2685.73  1013.6 2691.62
  1033.7 2691.82  1063.8 2690.88  1073.8 2692.12  1083.8 2695.22    1144 2718.37
#Mann= 3 , 0 , 0
       0     .06       0     547    .045       0     562     .06       0
Bank Sta=547,562
XS Rating Curve= 0 ,0
Exp/Cntr=0.3,0.1

Type RM Length L Ch R = 1 ,39618.4 ,345.2,352.3,359.4
XS GIS Cut Line= 2
     2073989.997       370863.01     2073927.812      371723.391
#Sta/Elev= 30
       0 2775.98    20.1 2771.34    60.2 2762.78   150.5 2742.34   210.6 2727.51
   230.7 2722.87   280.8 2713.03   300.9 2708.73     321 2703.63     341    2698
   391.2 2682.66   401.2 2680.55   461.4  2672.2   471.4 2671.29   481.5 2670.99
   506.6 2671.08   521.6 2671.37   621.9 2678.06     652 2679.77   692.1 2681.27
   732.2 2681.87   742.3 2682.78   762.3 2685.44   772.4 2686.02   792.4 2685.99
   822.5 2684.23   832.5 2684.39   842.6 2686.65   852.6 2692.51   862.6 2699.54
#Mann= 3 , 0 , 0
       0      .1       0   506.6    .045       0   521.6     .06       0
Bank Sta=506.6,521.6
XS Rating Curve= 0 ,0
Exp/Cntr=0.3,0.1

Type RM Length L Ch R = 1 ,39266.1 ,417.4,417.4,417.4
XS GIS Cut Line= 2
     2073809.474      370811.041     2073544.122      371469.196
#Sta/Elev= 30
       0 2747.88      50 2739.01      80 2734.51      90 2732.82   169.9  2717.9
   199.9 2712.99   209.9 2711.02   259.9 2699.44   299.8 2689.46   369.8 2674.85
   379.8 2673.34   409.8 2670.19   439.8    2668   469.8 2667.03   489.8 2666.14
   527.3 2665.87   539.7 2665.84   542.3 2665.86   549.7 2665.91   559.7 2666.42
   569.7 2667.44   609.7 2672.33   639.7 2677.02   649.7 2678.22   659.7 2678.52
   669.6 2678.08   679.6 2676.62   689.6 2675.51   699.6 2675.97   709.6 2679.22
#Mann= 3 , 0 , 0
       0      .1       0   527.3    .045       0   542.3      .1       0
Bank Sta=527.3,542.3
XS Rating Curve= 0 ,0
Exp/Cntr=0.3,0.1

Type RM Length L Ch R = 1 ,38848.7 ,440.9,433.3,425.7
XS GIS Cut Line= 2
     2073407.903      370695.437     2073162.134      371305.019
#Sta/Elev= 30
       0 2716.83    99.6 2698.12   119.5 2693.92   149.4 2687.06   169.3 2683.01
   179.2 2681.16   189.2 2679.48   199.2 2677.93   209.1 2676.71   219.1 2675.93
     249 2674.52   298.8 2670.73   368.5 2666.46   418.3 2663.65   448.1  2661.8
     478  2660.5     488 2660.31   496.7 2660.38   507.9 2660.92   511.7 2661.36
   517.8 2662.07   527.8 2663.64   557.7 2669.17   567.6 2670.77   577.6 2671.42
   597.5  2670.5   607.5 2671.43   617.4 2674.15   637.3  2680.5   657.3 2686.33
#Mann= 3 , 0 , 0
       0      .1       0   496.7    .045       0   511.7      .1       0
Bank Sta=496.7,511.7
XS Rating Curve= 0 ,0
Exp/Cntr=0.3,0.1

Type RM Length L Ch R = 1 ,38415.4 ,418.2,420.1,421.9
XS GIS Cut Line= 2
      2072860.24      370593.069     2072823.174      371268.893
#Sta/Elev= 30
       0 2700.94    49.8 2692.75    69.7 2689.17   109.5 2680.09   119.4 2677.99
   129.4 2676.26   159.3 2672.33     209 2666.32   238.9 2662.99   318.5  2655.3
   348.4 2652.86   392.7 2650.88   398.1  2650.7   407.7 2650.82     418 2651.69
     438 2654.26   457.9 2656.02   467.8 2656.69   487.7 2657.56   507.6 2658.13
   567.4 2659.21   577.3 2660.21   587.3 2661.74   597.2 2662.95   607.2 2663.38
   627.1 2663.29     637 2664.39     647 2668.01   656.9 2673.52   676.8  2684.1
#Mann= 3 , 0 , 0
       0      .1       0   392.7    .045       0   407.7      .1       0
Bank Sta=392.7,407.7
XS Rating Curve= 0 ,0
Exp/Cntr=0.3,0.1

Type RM Length L Ch R = 1 ,37995.3 ,317.8,324.7,331.8
XS GIS Cut Line= 2
     2072499.487      370576.103      2072411.52      371255.366
#Sta/Elev= 30
       0  2680.4    10.1 2679.24    40.3 2676.76    50.4  2675.7   120.9 2668.02
   161.2 2663.07   171.2 2662.03   181.3 2661.21   241.7 2657.65   261.9 2656.65
   322.3 2654.12   332.4 2653.82   362.6 2653.36   382.8  2652.6   392.8    2652
     413 2650.45   493.6 2643.23   503.6 2642.73   518.9 2642.68   533.9 2642.61
   543.9  2642.5     554 2643.03   564.1 2644.48   624.5 2656.95   634.6 2658.15
   644.6 2658.26   654.7 2657.77   664.8 2657.74   674.9 2659.13   684.9 2662.34
#Mann= 3 , 0 , 0
       0      .1       0   518.9    .045       0   533.9      .1       0
Bank Sta=518.9,533.9
XS Rating Curve= 0 ,0
Exp/Cntr=0.3,0.1

Type RM Length L Ch R = 1 ,37670.5 ,790,776.1,762.1
XS GIS Cut Line= 2
     2072367.072      370533.886     2072059.119       371178.42
#Sta/Elev= 30
       0 2686.36    40.2  2679.8   100.6 2670.97     161 2660.86   201.2  2656.1
   261.6 2649.97   281.7 2648.56   311.9 2648.62   392.4 2652.46   422.6 2652.36
   442.7 2651.06   472.9 2647.38   482.9 2645.16     503 2637.89   513.1 2637.41
   539.9  2637.6   554.9 2639.32   563.4 2641.72   583.5 2649.44   593.6 2652.32
   603.6 2653.68   623.8 2653.57   633.8 2654.43   643.9 2659.62     654 2669.42
     664 2680.02   674.1 2688.13   684.1 2693.76   694.2 2697.05   714.3 2700.77
#Mann= 3 , 0 , 0
       0      .1       0   539.9    .045       0   554.9      .1       0
Bank Sta=539.9,554.9
XS Rating Curve= 0 ,0
Exp/Cntr=0.3,0.1

Type RM Length L Ch R = 1 ,36894.1 ,733.7,728.6,723.6
XS GIS Cut Line= 2
     2071427.656      370209.564     2071615.652      371339.645
#Sta/Elev= 30
       0 2819.81    80.4  2786.7   160.8  2751.1     201 2730.73   281.4 2683.69
   311.5 2667.13   331.6 2656.42   371.8 2636.75   381.9 2632.74   391.9 2630.72
     402 2630.57   402.7 2630.58   417.7 2630.76   432.1 2631.43   482.4 2637.17
   502.5 2638.48   542.7  2638.5   653.2  2635.3   703.4 2637.05   773.8 2643.28
   793.9 2643.63     814 2642.82     824 2644.02   844.1 2649.61   854.2 2651.04
   994.9 2663.75    1015 2664.88    1025 2666.33  1035.1 2669.55  1145.6 2714.93
#Mann= 3 , 0 , 0
       0      .1       0   402.7    .045       0   417.7      .1       0
Bank Sta=402.7,417.7
XS Rating Curve= 0 ,0
Exp/Cntr=0.3,0.1

Type RM Length L Ch R = 1 ,36165.3 ,402.9,405.8,408.8
XS GIS Cut Line= 2
     2070628.344       370345.28     2071109.729      371460.358
#Sta/Elev= 30
       0 2877.98    30.1 2863.43    70.3 2841.43    90.3 2832.48   120.4    2823
   150.6 2815.94   170.6 2812.26   180.7 2808.84   200.8 2798.81   301.1 2745.38
   381.4 2697.52   441.6 2660.21   491.8  2631.4   511.9    2622     522 2619.44
   547.4 2618.48   562.1 2618.32   562.4 2618.32   582.2 2618.61   652.4 2624.71
   672.5 2624.37   702.6 2622.18   853.2 2632.97   883.3 2634.34   973.6 2650.24
   993.7 2651.89  1043.9  2654.2    1074  2658.2  1164.4 2679.25  1214.6 2692.53
#Mann= 3 , 0 , 0
       0      .1       0   547.4    .045       0   562.4      .1       0
Bank Sta=547.4,562.4
XS Rating Curve= 0 ,0
Exp/Cntr=0.3,0.1

Type RM Length L Ch R = 1 ,35759.5 ,491.3,493.5,495.7
XS GIS Cut Line= 2
     2070383.715      370545.856     2070704.999      371692.175
#Sta/Elev= 30
       0 2804.95    70.6 2774.13   131.2 2747.03   151.3 2737.66   242.1 2691.41
   363.2 2628.42   373.3  2623.5   383.4  2619.8   393.5 2618.08   403.6 2617.42
   534.7  2611.1     565 2610.17   587.7 2610.74   602.7 2611.34   625.5  2612.4
   635.6 2613.65   716.3 2627.25   726.4 2628.19   736.5  2628.7   746.6 2629.96
   756.7 2632.62   837.4  2660.4   847.5 2663.03   887.8 2672.19   958.4 2688.94
  1049.2 2709.42  1069.4 2714.29  1109.8 2725.28  1160.2  2740.3  1190.5 2748.74
#Mann= 3 , 0 , 0
       0      .1       0   587.7    .045       0   602.7      .1       0
Bank Sta=587.7,602.7
XS Rating Curve= 0 ,0
Exp/Cntr=0.3,0.1

Type RM Length L Ch R = 1 ,35266   ,484.3,491.1,497.9
XS GIS Cut Line= 2
      2069950.43      370441.886     2070150.263      371643.114
#Sta/Elev= 30
       0 2771.52    20.1 2766.55    90.6 2751.83   120.8 2745.06   191.2  2727.8
   211.3 2721.73   231.5 2714.88   261.7  2703.8   301.9 2688.16     322 2681.72
   362.3 2669.83   452.9 2639.27   483.1 2630.64   523.3 2621.32   553.5 2616.25
   573.6    2614   684.4 2610.44   724.6 2608.18   774.9 2603.64     785 2603.42
   822.7 2605.08   837.7    2607   875.6  2617.2   905.8 2621.75   915.8 2625.55
   956.1 2646.19   976.2 2654.42    1107 2701.33  1187.5 2728.02  1217.7 2737.53
#Mann= 3 , 0 , 0
       0      .1       0   822.7    .045       0   837.7      .1       0
Bank Sta=822.7,837.7
XS Rating Curve= 0 ,0
Exp/Cntr=0.3,0.1

Type RM Length L Ch R = 1 ,34774.9 ,484.9,484.8,484.7
XS GIS Cut Line= 2
     2069698.557      370546.134     2069535.273      371717.725
#Sta/Elev= 30
       0 2740.37    40.1 2723.05    90.2 2703.67   130.3 2687.46     391 2617.46
     411 2612.79   431.1 2609.86   521.3 2600.13   541.3 2598.71   551.4 2598.66
     584 2598.81     599 2599.02   621.5  2601.1   691.7 2611.18   701.7  2612.3
   721.8 2613.33   731.8 2615.27   741.8 2618.39   751.8 2622.68   781.9 2638.15
     812  2652.5     822 2657.04   852.1 2669.04   882.2 2679.54   942.3 2695.59
  1022.5 2719.56  1052.6 2727.99  1062.6 2731.38  1142.8 2765.61  1182.9 2784.36
#Mann= 3 , 0 , 0
       0      .1       0     584    .045       0     599      .1       0
Bank Sta=584,599
XS Rating Curve= 0 ,0
Exp/Cntr=0.3,0.1

Type RM Length L Ch R = 1 ,34290.1 ,627.3,627.3,627.3
XS GIS Cut Line= 2
     2069246.226       370405.57     2069086.203      371553.769
#Sta/Elev= 30
       0 2758.17    50.4  2739.9   201.6 2689.57   221.8 2684.23     252 2677.54
   332.7 2661.71   383.1 2648.62   413.3 2639.34   463.7 2621.12   473.8 2617.14
   514.1 2598.94   524.2 2595.67   534.3 2593.87   544.4 2593.37   572.1 2593.95
   587.1 2594.88   665.3 2600.08   786.3 2602.98   806.5 2604.35   826.6 2607.07
   856.9 2612.42   907.3 2623.53   937.5 2631.66   967.8  2640.8   987.9 2647.68
  1008.1 2655.77  1018.2 2660.86  1058.5  2683.8    1119 2713.66  1159.3 2734.94
#Mann= 3 , 0 , 0
       0      .1       0   572.1    .045       0   587.1      .1       0
Bank Sta=572.1,587.1
XS Rating Curve= 0 ,0
Exp/Cntr=0.3,0.1

Type RM Length L Ch R = 1 ,33662.8 ,307.3,308.3,309.2
XS GIS Cut Line= 2
     2068620.476      370419.083     2068463.704       371543.95
#Sta/Elev= 30
       0 2708.99    40.2 2689.53    60.3  2681.5   100.5 2667.91     201 2630.76
   221.1 2623.75   281.4 2604.36   301.5 2599.11   311.6    2597   331.7 2595.08
   412.1 2593.24   452.3 2591.31   482.4 2588.65   522.6 2582.55   542.7 2581.83
   560.4 2582.18   575.4  2583.9   613.1 2591.28   643.2 2596.45   663.4 2598.29
   693.5 2599.25   703.6 2600.76   844.3 2633.62   864.4 2638.74   884.5 2644.55
   934.7 2662.16  1045.3 2697.54  1055.3  2700.6  1095.5 2711.18  1135.7 2724.29
#Mann= 3 , 0 , 0
       0      .1       0   560.4    .045       0   575.4      .1       0
Bank Sta=560.4,575.4
XS Rating Curve= 0 ,0
Exp/Cntr=0.3,0.1

Type RM Length L Ch R = 1 ,33354.5 ,402.6,405.6,408.5
XS GIS Cut Line= 2
     2068329.608      370433.912     2068165.111      371333.505
#Sta/Elev= 30
       0 2650.94      10  2647.9    90.4 2629.91   150.7  2614.7   190.9 2604.91
   261.3 2589.89   281.4  2586.3   291.4 2585.27   301.5 2584.66   422.1 2578.42
   452.2 2577.43   472.3 2577.23     475 2577.23     490 2577.36   502.5 2578.28
   512.5 2580.31   532.6 2585.66   542.7 2587.93   582.9 2594.73   592.9 2596.04
     603 2596.33   633.1 2596.22   673.3 2597.82   693.4 2599.34   723.6 2602.89
   733.6 2604.37     804 2616.74   824.1 2620.72   884.4  2634.1   914.5 2641.83
#Mann= 3 , 0 , 0
       0      .1       0     475    .045       0     490      .1       0
Bank Sta=475,490
XS Rating Curve= 0 ,0
Exp/Cntr=0.3,0.1
